HEC-RAS study LAURELCK3.prj: LAURELCK3

--- LAURELCK3.g01 (geometry) --- (continued)

Type RM Length L Ch R = 1 ,29250.4 ,419.6,422.2,421.9
XS GIS Cut Line= 2
     2148519.318       243786.03      2149256.08      244285.162
#Sta/Elev= 30
       0    2569     9.8 2566.35    32.7 2550.24    81.8 2519.97     144 2486.86
     193 2463.48   202.8 2456.69   215.9 2454.68   245.4 2437.16   278.1 2424.37
   323.9 2403.93   346.8  2390.8   366.4 2388.26     409 2389.43   471.1 2388.32
   484.2 2383.84   490.8  2383.7   500.6 2383.87   503.8 2384.27   513.7 2389.36
   516.9 2389.51   634.7 2390.01  743.642393.254   765.6 2392.01  773.872393.088
   817.9 2417.47   837.6 2426.37     867 2437.88   883.4  2441.4   889.9 2444.77
#Mann= 5 ,-1 , 0
       0     .12       0   484.2    .045       0   500.6     .12       0
  743.64    .016       0  773.87     .12       0
#XS Ineff= 2 , 0
          466.46 2394.34  517.03         2394.76
Permanent Ineff=
       F       F
Bank Sta=484.2,500.6
XS Rating Curve= 0 ,0
Exp/Cntr=0.3,0.1

Type RM Length L Ch R = 1 ,28828.2 ,341.3,350,361.8
XS GIS Cut Line= 3
     2148333.053      244091.647     2148680.237      244378.447
     2149076.104      244652.557
#Sta/Elev= 30
       0 2549.18    16.3 2538.04    94.6 2491.64   104.4  2483.8   120.7 2479.33
   146.8 2462.96   218.6 2424.28     235 2419.94   244.7 2413.78   261.1 2406.11
   290.4 2382.43   293.7 2380.74   306.7 2379.59   336.1 2382.68   414.4 2384.38
   437.3 2382.46  444.862380.448   460.2 2380.56     506 2383.31   555.1 2381.78
   574.8 2382.44     601  2386.6  657.992386.713   669.8 2388.05   692.7 2387.52
  700.382391.124   771.3 2434.34   810.6 2456.42   866.3 2485.82   931.8 2515.69
#Mann= 5 ,-1 , 0
       0     .12       0  444.86    .045       0   460.2     .12       0
  657.99    .016       0  700.38     .12       0
Bank Sta=444.86,460.2
XS Rating Curve= 0 ,0
Exp/Cntr=0.3,0.1

Type RM Length L Ch R = 1 ,28478.2 ,414.5,403.8,389.5
XS GIS Cut Line= 3
     2148243.732      244193.305     2148499.205      244655.578
     2148681.617       245058.17
#Sta/Elev= 30
       0 2554.37    42.6 2527.67   111.5 2489.33   124.7 2478.57   141.1 2474.09
   226.4 2429.53   239.5 2426.77   272.3 2409.53   305.1 2379.58   324.8 2375.38
     351 2379.24   403.5 2377.98   423.2 2380.58   436.3 2380.32   449.4 2377.26
   501.9 2379.54   518.3 2377.19  532.332377.182   541.3 2379.65   583.8 2378.24
   616.6 2381.71   655.8  2379.6  725.852382.725   734.4 2384.44   760.6  2383.7
  775.052390.214   819.6 2406.53   881.8  2433.7   914.5 2443.49   970.2 2464.18
#Mann= 5 ,-1 , 0
       0     .12       0   518.3    .045       0  532.33     .12       0
  725.85    .016       0  775.05     .12       0
#XS Ineff= 2 , 0
                          630.55         2386.32
Permanent Ineff=
       F       F
Bank Sta=518.3,532.33
XS Rating Curve= 0 ,0
Exp/Cntr=0.3,0.1

Type RM Length L Ch R = 1 ,28074.4 ,302.7,303.1,301.5
XS GIS Cut Line= 2
     2147744.914      244524.496     2148624.323      245060.454
#Sta/Elev= 30
       0 2673.69    62.3 2676.13    88.6 2659.15   127.9 2642.28   147.6 2630.23
   229.6 2572.24   268.9 2537.06   341.1  2479.4   347.7 2471.44   364.1 2465.75
     387 2445.99   419.8 2423.18   429.6 2414.12   439.5 2397.89     446 2390.64
   465.7 2372.13   475.6 2369.18   482.1 2368.55   488.7 2369.34   521.5 2374.31
   577.2  2377.4   665.8 2377.77   678.9 2376.01   698.6 2378.55   800.3 2377.86
  877.642382.674   911.8 2383.84  919.182388.776   934.8 2394.69  1029.9  2441.8
#Mann= 5 ,-1 , 0
       0     .12       0   475.6    .045       0   488.7     .12       0
  877.64    .016       0  919.18     .12       0
#XS Ineff= 2 , 0
                           598.8          2379.4
Permanent Ineff=
       F       F
Bank Sta=475.6,488.7
XS Rating Curve= 0 ,0
Exp/Cntr=0.3,0.1

Type RM Length L Ch R = 1 ,27771.3 ,351,353.3,354.3
XS GIS Cut Line= 3
     2147612.508       244784.47     2148001.461      245020.569
     2148389.703      245257.829
#Sta/Elev= 30
       0  2642.3    45.8 2643.23    68.7 2641.76    85.1  2637.8   104.8 2628.07
   193.1  2573.4   219.3 2555.18   258.6 2524.34   284.8 2499.55   314.2 2475.62
   337.2 2458.82   356.8 2441.99     383 2417.74   405.9 2390.53   425.5 2370.01
   435.4 2366.94   464.8 2366.38   474.6 2365.88  479.922366.435   487.7 2368.89
   510.6 2369.91   533.6 2373.33   618.7 2372.22   739.8 2378.09     802 2384.43
   818.4 2387.41  827.562390.878   854.4 2391.18  869.062398.947     910 2409.42
#Mann= 5 ,-1 , 0
       0     .12       0   464.8    .045       0  479.92     .12       0
  827.56    .016       0  869.06     .12       0
#XS Ineff= 2 , 0
                          544.62         2377.36
Permanent Ineff=
       F       F
Bank Sta=464.8,479.92
XS Rating Curve= 0 ,0
Exp/Cntr=0.3,0.1

Type RM Length L Ch R = 1 ,27418   ,345.3,350,355.8
XS GIS Cut Line= 3
     2147441.441      245041.086     2147809.534      245312.047
     2148180.666       245575.65
#Sta/Elev= 30
       0 2593.06    13.1 2593.82    32.6 2592.12    65.3 2583.96    94.7 2571.79
   163.2 2537.32   202.4 2516.39   218.7 2504.75   241.6 2491.47   280.8 2463.32
   329.7 2423.37   359.1 2403.51   378.7  2387.5   404.8  2370.8   414.6 2366.52
   427.7 2367.22   450.5 2362.61   457.1 2361.93   464.6 2362.56   489.8 2364.52
   509.5 2369.53   584.8 2366.63   643.7 2366.93   679.8 2369.09     706 2368.23
  738.322374.489   771.5 2375.22  777.682379.084     814 2396.17   912.3  2451.3
#Mann= 5 ,-1 , 0
       0     .12       0   450.5    .045       0   464.6     .12       0
  738.32    .016       0  777.68     .12       0
#XS Ineff= 2 , 0
                          507.55         2371.43
Permanent Ineff=
       F       F
Bank Sta=450.5,464.6
XS Rating Curve= 0 ,0
Exp/Cntr=0.3,0.1

Type RM Length L Ch R = 1 ,27068   ,338,350,363.4
XS GIS Cut Line= 3
     2147314.201      245247.906     2147657.156      245622.321
     2147939.758      245966.672
#Sta/Elev= 30
       0 2486.79    16.4 2479.79      59 2473.72    78.6 2468.54   101.6 2460.08
   144.1 2437.68   199.8 2401.44   216.2 2389.27   229.3 2376.88   255.5 2363.48
   281.7 2359.83   363.6 2363.98   402.9 2361.69   419.3 2363.23   458.6  2363.2
   497.9 2359.02   504.5 2358.66     511 2358.97   517.6 2360.44   520.8 2362.61
   523.62366.233   527.4 2369.59   543.8 2370.81   553.6  2378.6  564.512385.272
     642 2422.32   684.6 2437.28   756.7 2454.18   884.4 2473.05   953.2 2481.42
#Mann= 5 ,-1 , 0
       0     .12       0   497.9    .045       0     511     .12       0
   523.6    .016       0  564.51     .12       0
Bank Sta=497.9,511
XS Rating Curve= 0 ,0
Exp/Cntr=0.3,0.1

Type RM Length L Ch R = 1 ,26718   ,341.8,350,352.9
XS GIS Cut Line= 3
       2147222.6      245287.473     2147331.185      245732.875
     2147371.573      246186.182
#Sta/Elev= 30
       0 2478.75    42.6 2454.49    68.8 2435.35    91.7  2422.3   160.5 2393.78
   229.2 2356.12   248.9 2358.06   311.1 2356.87   324.2 2359.43   350.4 2359.14
   366.8 2356.77   412.6    2359     429  2355.9   448.6 2354.41   455.2 2353.97
   461.7 2354.28   481.4 2357.69   504.3 2374.61  521.252382.202   530.5 2387.39
   550.1 2389.26   556.7 2395.19     5612397.163   599.2 2412.04   684.4 2437.66
   723.6 2451.17   782.6 2465.24   844.8 2475.81   897.2 2482.26   913.6 2482.18
#Mann= 5 ,-1 , 0
       0     .12       0   448.6    .045       0   461.7     .12       0
  521.25    .016       0     561     .12       0
Bank Sta=448.6,461.7
XS Rating Curve= 0 ,0
Exp/Cntr=0.3,0.1

Type RM Length L Ch R = 1 ,26368   ,338.3,350,361
XS GIS Cut Line= 3
     2147040.005      245313.384     2146986.956      245783.622
     2146963.209      246234.782
#Sta/Elev= 30
       0 2435.32    39.2 2411.45    71.8 2388.14    91.4 2370.55   104.4 2356.13
     111 2351.98   133.8 2350.52   150.1 2353.71   176.2 2353.96   199.1 2352.03
   225.2 2354.13   290.5 2352.36   336.2  2355.3   398.2 2356.23   453.6  2350.5
   463.4 2350.69   473.2 2350.35  478.442350.697     483 2352.22   499.4 2370.76
   515.8 2381.04   558.3 2389.07  568.042393.028   591.1 2393.39  605.382400.368
   636.9 2407.02   679.5  2412.3   777.7 2429.66   849.7 2447.64     925 2453.42
#Mann= 5 ,-1 , 0
       0     .12       0   463.4    .045       0  478.44     .12       0
  568.04    .016       0  605.38     .12       0
Bank Sta=463.4,478.44
XS Rating Curve= 0 ,0
Exp/Cntr=0.3,0.1

Type RM Length L Ch R = 1 ,26018   ,338.5,350,363.2
XS GIS Cut Line= 3
     2146944.529      245280.962     2146655.736      245684.707
     2146423.393      246067.392
#Sta/Elev= 30
       0 2423.28    16.3 2411.67    55.5 2388.37    88.2 2362.24   101.2 2353.07
   107.8 2350.24   179.6  2346.3   202.5 2349.64   313.5 2351.93   346.2 2350.34
   382.1 2351.14     405 2349.15   440.9 2351.02     467 2345.67   483.3 2346.53
  497.892346.531   509.5  2351.8   525.8 2366.65   535.6  2373.5  553.872383.423
   571.6 2384.51   581.4 2390.93  591.712395.121   663.1 2419.29   685.9 2428.52
   702.3 2436.81   712.1 2439.12     748 2457.37   819.9  2489.9   944.1 2540.51
#Mann= 5 ,-1 , 0
       0     .12       0   483.3    .045       0  497.89     .12       0
  553.87    .016       0  591.71     .12       0
Bank Sta=483.3,497.89
XS Rating Curve= 0 ,0
Exp/Cntr=0.3,0.1

Type RM Length L Ch R = 1 ,25668   ,363.4,350,339.2
XS GIS Cut Line= 3
     2146882.333      245202.822     2146448.941      245410.984
     2146038.576      245596.918
#Sta/Elev= 30
       0 2442.46    42.5 2419.14    98.1 2395.01   117.7 2384.65   147.2 2372.76
   176.6 2355.53   196.2 2346.98     206 2345.73   258.4 2346.22   297.6 2342.21
   330.3  2346.3   353.2 2347.27   392.5 2346.17   415.4 2342.27   441.5 2345.35
     471 2339.29   484.1 2338.83   488.3 2339.31   510.2  2347.6  560.522350.653
  618.032350.201   683.2 2349.65   709.3 2352.34   725.6 2358.08   748.5 2369.21
  768.822373.115   797.5 2372.12  813.86 2374.32   885.6 2372.66   931.3    2375
#Mann= 7 ,-1 , 0
       0     .12       0     471    .045       0   488.3     .12       0
  560.52     .06       0  618.03     .12       0  768.82    .016       0
  813.86     .12       0
Bank Sta=471,488.3
XS Rating Curve= 0 ,0
Exp/Cntr=0.3,0.1

Type RM Length L Ch R = 1 ,25318   ,344.9,350,350.5
XS GIS Cut Line= 3
     2146497.113       244740.53     2146276.269      245133.139
     2145974.541       245507.39
#Sta/Elev= 30
       0 2401.08    65.3 2390.75     124 2385.36     173  2378.8   257.9 2361.66
   323.2 2351.68   336.2 2347.66   372.1 2345.27   391.7 2337.39   417.8 2337.22
   440.7 2332.38   443.9 2332.24   453.7 2332.37   460.3 2332.69   515.9 2344.25
  630.532349.658  683.71 2351.85   692.5 2352.43   702.3 2350.59   721.9 2350.16
   748.1 2353.34  808.042356.049   816.7 2356.26   829.8 2359.03   833.1 2358.98
   839.6 2355.97  847.74 2357.37   878.9 2359.68   898.5 2359.03   931.2 2361.72
#Mann= 7 ,-1 , 0
       0     .12       0   440.7    .045       0   453.7     .12       0
  630.53    .016       0  683.71     .12       0  808.04    .016       0
  847.74     .12       0
Bank Sta=440.7,453.7
XS Rating Curve= 0 ,0
Exp/Cntr=0.3,0.1

Type RM Length L Ch R = 1 ,24968   ,286.2,282.5,276.9
XS GIS Cut Line= 3
     2146293.004      244594.917     2146006.423      244944.117
     2145698.536      245302.088
#Sta/Elev= 30
       0 2387.59    98.2 2360.26   117.8 2353.29   134.2 2349.96   212.8 2345.95
   248.8 2347.63   268.4 2342.22   297.9 2341.19   314.2 2336.05   350.3 2336.43
   373.2 2333.62   412.5  2332.8   441.9 2328.25   451.7 2327.68  455.682328.308
   517.3  2341.4   612.4 2342.53  625.792346.068   635.4 2350.11   651.8 2352.01
  667.732361.344   697.7 2375.54   743.6 2401.15   753.4 2407.36   763.2 2415.73
   776.4 2419.28   789.5 2429.49   858.3 2468.44   891.1 2483.24   923.9 2494.78
#Mann= 5 ,-1 , 0
       0     .12       0   441.9    .045       0  455.68     .12       0
  625.79    .016       0  667.73     .12       0
Bank Sta=441.9,455.68
XS Rating Curve= 0 ,0
Exp/Cntr=0.3,0.1

Type RM Length L Ch R = 1 ,24685.5 ,345.8,348.1,349.4
XS GIS Cut Line= 2
     2145988.284      244417.304     2145559.518      245202.647
#Sta/Elev= 30
       0 2379.62     154 2344.67   216.3 2340.69   245.8 2336.04   268.8 2336.87
   275.3 2335.02   285.1 2329.64   291.7 2328.11   383.5 2330.35  398.342325.776
   399.7  2325.6   416.2 2325.75   468.7 2327.32   485.1 2325.92   488.4 2326.52
   494.9 2333.43   501.5 2336.74  540.392338.678   560.5 2339.83  568.242343.218
   609.6 2373.68   698.1 2430.94     708 2438.63   721.1 2442.49   730.9 2450.32
   757.1 2463.63   819.4 2500.16   845.6 2514.03     862 2521.92   894.8 2533.54
#Mann= 5 ,-1 , 0
       0     .12       0  398.34    .045       0   416.2     .12       0
  540.39    .016       0  568.24     .12       0
Bank Sta=398.34,416.2
XS Rating Curve= 0 ,0
Exp/Cntr=0.3,0.1

Type RM Length L Ch R = 1 ,24337.4 ,427.6,422.3,414.7
XS GIS Cut Line= 3
     2145738.613      244250.597     2145484.128      244627.967
     2145238.873      245011.176
#Sta/Elev= 30
       0 2387.31   117.9 2369.93   183.4 2366.33   219.4 2363.13   225.9 2359.72
   245.6  2343.7   265.2 2329.26   271.8 2325.78   275.1 2325.24   320.9  2324.8
   350.4  2326.5     370 2325.03   412.6 2326.55   442.1 2322.02   451.9 2321.67
   467.4 2321.82   471.5 2322.43   487.9 2329.02  535.322327.967  570.892329.413
   586.1 2327.64   595.9 2330.02   618.8 2341.69   651.6 2356.28   703.9 2383.09
   769.4 2414.61     861 2465.08   893.8 2480.88   900.3 2483.15   910.1 2483.83
#Mann= 5 ,-1 , 0
       0     .12       0   451.9    .045       0   467.4     .12       0
  535.32    .016       0  570.89     .12       0
#XS Ineff= 2 , 0
          347.47 2328.32
Permanent Ineff=
       F       F
Bank Sta=451.9,467.4
XS Rating Curve= 0 ,0
Exp/Cntr=0.3,0.1

Type RM Length L Ch R = 1 ,23915.1 ,355.6,350.6,343.7
XS GIS Cut Line= 3
      2145293.26       243966.55     2145150.462      244399.114
     2144985.323      244838.955
#Sta/Elev= 30
       0 2460.18    16.4  2457.4    91.8 2455.76   131.1 2445.92   173.7 2438.96
   196.6 2432.31   216.3 2423.68   321.2 2360.61   334.3 2354.01   363.8 2343.14
   393.3 2337.11   409.6 2336.07   419.5 2333.77     426  2329.7   435.9 2318.31
  441.632315.983   445.7 2315.81   455.5 2315.84   501.2 2321.12   566.4 2319.96
   595.8 2323.27  655.272324.484   674.1 2321.88  690.42 2324.85   729.6 2325.48
   749.2 2335.04   775.3 2344.01   791.6 2351.45   876.4 2397.78   925.3 2420.61
#Mann= 5 ,-1 , 0
       0     .12       0  441.63    .045       0   455.5     .12       0
  655.27    .016       0  690.42     .12       0
#XS Ineff= 2 , 0
                          652.44         2326.69
Permanent Ineff=
       F       F
Bank Sta=441.63,455.5
XS Rating Curve= 0 ,0
Exp/Cntr=0.3,0.1

Type RM Length L Ch R = 1 ,23564.5 ,340.8,352.7,366.1
XS GIS Cut Line= 3
     2144852.001      243893.172     2144808.711      244346.694
     2144774.377      244800.306
#Sta/Elev= 30
       0  2452.1   196.6 2418.72   229.4 2411.57   245.8 2405.08   291.7 2379.66
   311.4    2367   357.3 2340.87   376.9 2326.52   383.5 2324.37   393.3 2317.96
   399.9 2315.85     413 2315.97  443.992311.928   455.6 2311.75   458.9 2311.84
     485 2315.14     508 2312.58     521 2318.59   524.3 2318.76   537.4 2317.81
   553.8 2319.26   563.6 2318.14   583.2 2320.32     593  2318.7  645.812321.221
   668.3 2321.76  679.982325.746   782.9 2376.54     845 2414.68   910.5 2449.19
#Mann= 5 ,-1 , 0
       0     .12       0  443.99    .045       0   458.9     .12       0
  645.81    .016       0  679.98     .12       0
Bank Sta=443.99,458.9
XS Rating Curve= 0 ,0
Exp/Cntr=0.3,0.1

Type RM Length L Ch R = 1 ,23211.8 ,340.9,350.6,351.4
XS GIS Cut Line= 3
     2144759.911      243861.716     2144500.448      244243.461
     2144184.043      244572.994
#Sta/Elev= 30
       0  2431.7    45.8 2418.29   121.1 2403.54   153.9 2391.23   229.2 2369.74
   278.2 2347.48   297.9 2332.31   320.8 2317.48     347 2317.99   373.2 2308.02
   389.6 2309.38   409.2 2307.87   428.8 2309.88   445.2 2306.79   448.5 2306.71
   458.3  2306.8   477.9 2308.54   500.7 2327.77     517 2338.78  550.242355.647
     566 2356.22     579 2364.77  592.19  2368.6   673.7 2382.43     690 2390.73
   738.9 2420.97   755.3 2427.96   804.2 2442.38   846.6 2445.04   918.4 2443.59
#Mann= 5 ,-1 , 0
       0     .12       0   445.2    .045       0   458.3     .12       0
  550.24    .016       0  592.19     .12       0
Bank Sta=445.2,458.3
XS Rating Curve= 0 ,0
Exp/Cntr=0.3,0.1

Type RM Length L Ch R = 1 ,22861.2 ,371.3,382,398
XS GIS Cut Line= 3
     2144650.411      243741.205     2144267.927      243985.647
     2143947.399       244321.91
#Sta/Elev= 30
       0 2406.38    39.2 2397.07    71.8  2387.1   182.9 2366.95   264.5  2347.2
   287.4 2339.18   297.2 2333.39   316.8  2330.4   329.8 2320.47   346.2 2312.74
   375.6 2304.37   395.1  2301.8   434.3 2305.11   446.4 2302.15   460.5 2302.16
   486.6 2303.76   493.2 2306.24   509.5 2317.07   558.6 2341.97  626.762379.774
   637.1 2386.78   656.8 2387.31  668.892390.219   679.7 2392.14   712.4 2406.02
   738.5 2411.29   774.5 2426.82   830.2 2435.92   879.2 2439.54   918.5 2444.79
#Mann= 5 ,-1 , 0
       0     .12       0   446.4    .045       0   460.5     .12       0
  626.76    .016       0  668.89     .12       0
Bank Sta=446.4,460.5
XS Rating Curve= 0 ,0
Exp/Cntr=0.3,0.1

Type RM Length L Ch R = 1 ,22479.2 ,307.3,318,332.6
XS GIS Cut Line= 3
     2144611.315      243624.324     2144081.715      243678.928
     2143642.093      243716.868
#Sta/Elev= 30
       0 2400.17    65.3 2377.31   107.8 2372.37   182.9 2355.45   192.7 2350.92
   215.6    2349   320.1  2320.2     343 2312.03   365.8 2296.15   382.2  2296.7
   398.5 2300.32   467.1 2301.27   493.2 2303.94   528.5 2298.22   543.5 2298.36
   571.6 2298.09   591.2 2305.88   610.8 2305.49   630.5 2310.35   659.9    2331
   676.2 2347.78   692.6 2361.93   741.6 2395.76   774.3 2412.18   800.4 2422.72
   823.3 2428.65   872.3 2434.49   898.5 2434.84   950.8 2431.07   973.7 2431.97
#Mann= 3 ,-1 , 0
       0     .12       0   528.5    .045       0   543.5     .12       0
Bank Sta=528.5,543.5
XS Rating Curve= 0 ,0
Exp/Cntr=0.3,0.1

Type RM Length L Ch R = 1 ,22161.2 ,351.9,350,349
XS GIS Cut Line= 3
     2144627.337      243561.344     2144162.056      243379.401
     2143783.845      243141.103
#Sta/Elev= 30
       0 2408.24    35.9 2399.26    75.1 2385.15   130.6 2375.02   140.4 2370.88
   176.3 2368.41     209 2353.62   284.1  2334.5   306.9 2326.14   323.3 2315.62
   339.6 2301.89   349.4 2297.14     369 2296.89   391.8 2292.54     418  2295.9
   463.7 2295.87   492.1 2292.33   499.6 2292.01   507.1 2292.43   532.2 2295.78
   571.4 2295.57     591 2303.14   626.8 2306.21     666 2316.67   705.2 2322.23
   731.3 2330.46   780.2  2358.5     865 2388.03   897.7 2405.71   946.6 2421.07
#Mann= 3 ,-1 , 0
       0     .12       0   492.1    .045       0   507.1     .12       0
#XS Ineff= 2 , 0
          366.97  2298.5  553.03         2298.41
Permanent Ineff=
       F       F
Bank Sta=492.1,507.1
XS Rating Curve= 0 ,0
Exp/Cntr=0.3,0.1

Type RM Length L Ch R = 1 ,21811.2 ,350,349.8,342.1
XS GIS Cut Line= 3
     2144822.357      243266.046      2144393.65      243135.999
     2143973.691      242875.931
#Sta/Elev= 30
       0 2494.74    42.5 2482.47    78.5 2467.71   117.7 2454.61   176.6 2429.78
   222.4 2413.65   238.7 2403.66   251.8 2400.09   271.4    2389   310.7 2376.12
   359.7  2352.2   372.8 2344.03   421.8 2297.69   434.9 2287.25   440.5  2284.8
     448 2283.83   455.5  2284.8   480.7 2286.93   500.3 2291.06   549.4 2288.08
   565.8 2290.58   582.1 2289.13   595.2 2294.99   631.2 2293.07   667.2  2295.4
   716.2 2293.27   791.5 2298.89   843.8 2307.73   886.4 2320.06     942 2341.83
#Mann= 3 ,-1 , 0
       0     .12       0   440.5    .045       0   455.5     .12       0
#XS Ineff= 2 , 0
                          508.77         2296.88
Permanent Ineff=
       F       F
Bank Sta=440.5,455.5
XS Rating Curve= 0 ,0
Exp/Cntr=0.3,0.1

Type RM Length L Ch R = 1 ,21461.4 ,349,349.4,347.7
XS GIS Cut Line= 3
     2144903.693       242917.19     2144455.741      242793.894
     2144014.657       242689.49
#Sta/Elev= 30
       0 2487.29     3.3  2485.6    16.4 2482.52    55.6 2465.42    68.7 2458.67
    98.2 2446.11     157 2417.66   235.6 2384.28   320.6 2341.96   369.7 2320.64
   389.4 2313.59     409 2300.91   428.6 2283.97   448.2  2278.6   461.3 2278.41
   464.6 2278.46   484.2 2279.22   503.7 2286.48   536.4 2284.81   559.2 2288.49
   630.9 2286.48   663.5 2289.82     719  2288.8   741.8 2291.63   803.8 2296.02
   816.8 2298.35   839.6 2304.76     869 2315.66   901.6 2332.74   917.9 2342.37
#Mann= 3 ,-1 , 0
       0     .12       0   448.2    .045       0   464.6     .12       0
#XS Ineff= 2 , 0
                          504.64          2293.5
Permanent Ineff=
       F       F
Bank Sta=448.2,464.6
XS Rating Curve= 0 ,0
Exp/Cntr=0.3,0.1

Type RM Length L Ch R = 1 ,21112   ,289.8,298.7,308.7
XS GIS Cut Line= 3
     2145028.627      242594.327     2144585.757      242473.337
     2144138.998      242391.038
#Sta/Elev= 30
       0 2423.08   147.6  2367.5   249.2 2326.72   301.7 2309.71   321.4 2301.22
   357.4 2283.33   383.7 2280.74   396.8 2281.85   429.6 2281.09   449.3 2275.51
   455.8 2275.19   465.6 2275.39   485.2  2277.1     495 2276.88   521.2 2279.85
   534.3 2279.57   547.3 2280.72   583.3  2277.8   599.6 2279.99   622.5 2278.02
   635.6  2280.5   684.6 2281.06   697.7 2280.28   710.8 2281.64   743.4 2280.35
   779.4  2282.3   789.2 2285.64   815.3 2299.98   854.6 2317.15   913.4 2348.35
#Mann= 3 ,-1 , 0
       0     .12       0   449.3    .045       0   465.6     .12       0
#XS Ineff= 2 , 0
          426.21 2284.32  639.83         2284.93
Permanent Ineff=
       F       F
Bank Sta=449.3,465.6
XS Rating Curve= 0 ,0
Exp/Cntr=0.3,0.1

Type RM Length L Ch R = 1 ,20813.3 ,391.7,404.8,417.6
XS GIS Cut Line= 3
     2145069.499      242496.605      2144579.48      242129.091
     2144505.102      241875.332
#Sta/Elev= 30
       0 2394.01   101.5 2350.92   160.5 2328.46   206.4 2309.38   229.3  2298.8
   258.8 2281.68   275.1 2275.29     285 2274.31   307.9 2274.79     357 2277.55
   376.7 2273.62   406.2 2272.83   432.4 2274.28   465.1 2272.97   478.2 2273.46
     511  2268.2   520.8 2267.51  526.152268.137   540.5 2270.34     547 2272.72
   576.5 2295.67   586.3 2302.19   645.2 2329.09   681.1 2347.24   700.7 2358.99
   736.6 2382.64   749.6 2392.47   759.4 2397.57   811.7 2433.43     877 2480.96
#Mann= 3 ,-1 , 0
       0     .12       0     511    .045       0  526.15     .12       0
#XS Ineff= 2 , 0
           358.1 2283.78
Permanent Ineff=
       F       F
Bank Sta=511,526.15
XS Rating Curve= 0 ,0
Exp/Cntr=0.3,0.1

Type RM Length L Ch R = 1 ,20408.6 ,620.6,589.1,556.7
XS GIS Cut Line= 3
     2145170.128       242428.79     2144988.558      241938.772
     2144564.167      241800.954
#Sta/Elev= 30
       0 2368.41    58.8 2343.04    91.4 2325.28     111 2318.82   140.4 2312.04
   169.8 2297.93     209 2281.82   228.6 2279.19   254.8 2273.54   267.8 2273.63
   310.3 2269.49   326.6 2270.84   395.2 2268.94   401.7 2268.12  419.582262.711
   424.6  2262.2   434.4 2262.64     454 2263.41     467 2267.23   489.9 2290.01
   522.6 2316.13     578 2348.29   600.7  2366.8   652.9 2389.43   786.4 2456.06
   802.7 2462.67   828.7  2475.6   903.6    2499   929.7 2509.41   968.8 2519.57
#Mann= 3 ,-1 , 0
       0     .12       0  419.58    .045       0   434.4     .12       0
Bank Sta=419.58,434.4
XS Rating Curve= 0 ,0
Exp/Cntr=0.3,0.1

Type RM Length L Ch R = 1 ,19819.5 ,344.1,320.8,296.5
XS GIS Cut Line= 2
     2145808.902      241551.569     2144581.668      241785.641
#Sta/Elev= 30
       0 2389.16    55.8 2370.54     141 2334.22   229.5 2303.11   275.4 2260.89
   288.6 2255.68     305 2253.88   337.8  2257.9   396.8 2253.55   419.7 2256.68
   455.8 2256.32   488.6 2252.24   501.7 2251.42     505 2252.24   511.6  2255.3
   524.7 2256.31   527.9 2258.86   541.1 2278.86   547.6 2285.35   573.8 2302.28
   590.2 2309.97   652.6 2326.12   724.7 2355.26     810 2385.43   836.2 2392.82
   964.1 2418.73  1052.6 2442.94  1157.5 2481.93  1216.6 2508.85  1249.4 2519.53
#Mann= 3 ,-1 , 0
       0     .12       0   488.6    .045       0     505     .12       0
Bank Sta=488.6,505
XS Rating Curve= 0 ,0
Exp/Cntr=0.3,0.1

Type RM Length L Ch R = 1 ,19498.7 ,475.7,486.6,497.1
XS GIS Cut Line= 3
     2145233.568      241074.676     2145043.248      241617.197
     2144472.288      241735.326
#Sta/Elev= 30
       0 2301.27    19.6 2295.65    45.7 2302.88    62.1 2304.35    81.7 2304.74
   101.3 2301.56   120.9 2289.82   150.3    2264   160.1 2257.94   166.6 2256.09
   235.2 2252.32   267.9 2253.76   333.2 2252.99   372.4    2247   398.5 2249.19
   423.1 2245.25   427.9 2244.99   438.1 2245.28   450.8 2248.57   473.7  2264.6
   525.9 2305.11   574.9 2335.29   728.9 2367.03   751.8 2374.96   781.3 2381.23
   866.5 2406.95   945.1 2437.59  1066.3 2494.51  1085.9  2505.5    1158 2535.54
#Mann= 3 ,-1 , 0
       0     .12       0   423.1    .045       0   438.1     .12       0
Bank Sta=423.1,438.1
XS Rating Curve= 0 ,0
Exp/Cntr=0.3,0.1

Type RM Length L Ch R = 1 ,19012   ,342,350,350.3
XS GIS Cut Line= 3
     2145002.143      240954.884     2144639.584       241305.72
     2144314.055        241611.2
#Sta/Elev= 30
       0 2335.75    52.4    2320   163.8 2290.05   176.9 2288.58   235.9 2274.64
     249 2269.56   288.3  2250.1   324.3 2240.58   347.3 2237.08     380 2240.88
   406.2 2240.25   458.6 2243.02   471.8 2242.24   481.6 2237.38   494.7 2236.25
   504.5 2235.63  509.152236.313   514.3 2238.17   524.1 2248.43   550.1  2269.3
   582.7 2303.09   608.8  2324.3   621.8 2333.34   647.9 2356.29   706.5 2399.31
   768.4 2441.34   817.3 2471.53   849.9 2487.49     889 2501.79   950.9  2519.9
#Mann= 3 ,-1 , 0
       0     .12       0   494.7    .045       0  509.15     .12       0
Bank Sta=494.7,509.15
XS Rating Curve= 0 ,0
Exp/Cntr=0.3,0.1

Type RM Length L Ch R = 1 ,18662   ,373.9,350,340.5
XS GIS Cut Line= 3
       2144921.4      240800.162     2144513.308      240983.386
     2144137.215      241310.471
#Sta/Elev= 30
       0 2374.11    45.7 2356.88   117.6 2326.22   173.1 2298.98   189.4 2290.02
   267.8 2255.59   280.8 2248.87   297.1 2236.76   300.4 2235.22   323.3 2231.35
   359.2 2237.11   372.2 2236.67   385.3 2238.35   408.2  2237.9   424.5 2237.07
   434.3 2232.04  442.742230.212   447.3    2230   457.2 2230.19   470.3 2230.62
   483.4  2233.6   509.6  2235.9   516.2  2239.3   529.3 2248.92   545.7 2256.92
   627.7 2284.67   670.3 2295.97     749  2312.2   844.1 2340.97   945.8 2368.61
#Mann= 3 ,-1 , 0
       0     .12       0  442.74    .045       0   457.2     .12       0
Bank Sta=442.74,457.2
XS Rating Curve= 0 ,0
Exp/Cntr=0.3,0.1

Type RM Length L Ch R = 1 ,18312   ,307.8,300.6,286.5
XS GIS Cut Line= 3
     2144325.662      240316.555     2144284.823      240754.517
     2144068.364      241250.739
#Sta/Elev= 30
       0 2432.29    81.5 2425.15   140.1  2408.3   159.6 2400.55     202 2375.59
   237.8 2342.31   267.2 2317.41   280.2 2303.44     290 2289.83   299.8 2273.96
   342.1 2235.32   358.4    2226   364.9 2224.13     417 2228.58   430.1 2224.01
   436.6 2223.44   446.4 2224.05   469.2  2224.5     479 2227.42   521.4 2228.02
   534.4 2231.93   544.2 2232.48   589.9  2231.2   661.6 2233.59   674.7 2236.84
   730.1 2257.68   821.4 2283.37   880.1 2302.11   942.1 2324.92   981.2 2336.67
#Mann= 3 ,-1 , 0
       0     .12       0   430.1    .045       0   446.4     .12       0
#XS Ineff= 2 , 0
                          506.23         2230.26
Permanent Ineff=
       F       F
Bank Sta=430.1,446.4
XS Rating Curve= 0 ,0
Exp/Cntr=0.3,0.1

Type RM Length L Ch R = 1 ,18011.4 ,387.9,399.4,405.4
XS GIS Cut Line= 3
     2143901.828      240321.433     2144007.064      240765.806
     2144025.254      241239.776
#Sta/Elev= 30
       0 2308.33    19.6 2302.89    48.9 2309.24   104.4 2324.46     124 2325.17
     137 2322.97   153.3 2317.58   169.6 2307.97   185.9 2300.57     212 2283.75
   238.1 2272.25     287 2241.56   313.1 2228.13   329.4 2224.43   352.3 2225.76
   391.4 2222.57   407.7 2223.05   430.6 2217.56   437.1 2216.99   443.6 2217.43
   492.6 2220.06   505.7 2218.36   551.5 2227.94   607.1 2226.91   649.7 2231.66
   751.1 2262.85   790.3 2278.28   806.7 2283.01   875.4  2310.8     931 2330.47
#Mann= 3 ,-1 , 0
       0     .12       0   430.6    .045       0   443.6     .12       0
#XS Ineff= 2 , 0
          407.64 2226.96  492.26         2227.67
Permanent Ineff=
       F       F
Bank Sta=430.6,443.6
XS Rating Curve= 0 ,0
Exp/Cntr=0.3,0.1

Type RM Length L Ch R = 1 ,17612   ,339.9,351,367.5
XS GIS Cut Line= 3
     2143753.691      240330.581     2143619.141      240830.397
     2143574.349      241271.937
#Sta/Elev= 30
       0 2278.02    91.7 2256.26   124.5 2243.34   144.1 2233.22   163.8 2228.55
   176.9 2223.17   229.3 2218.08   298.1 2220.02   317.8 2215.96   366.9 2219.42
   412.8 2215.58   432.4 2208.99   448.8 2213.68   481.6 2215.19   507.8 2208.79
   514.3 2208.57   520.9 2208.77   527.4 2211.62   537.2 2223.07   543.7 2227.27
   566.6 2232.46   644.9 2255.71   759.1 2270.26   811.3 2282.42   821.1 2282.73
   850.5 2277.73   883.1 2283.34   909.2 2297.39   928.8 2311.16   961.4 2327.42
#Mann= 3 ,-1 , 0
       0     .12       0   507.8    .045       0   520.9     .12       0
Bank Sta=507.8,520.9
XS Rating Curve= 0 ,0
Exp/Cntr=0.3,0.1

Type RM Length L Ch R = 1 ,17261   ,345.6,347.1,345.7
XS GIS Cut Line= 3
     2143671.134      240276.196     2143345.441      240622.087
     2142987.609      240897.344
#Sta/Elev= 30
       0 2277.28    72.1 2256.25    98.3  2247.2   127.8 2233.23   144.2 2222.09
   167.1 2214.43   235.9 2214.18   252.3 2216.14   281.8 2216.47   324.4  2214.9
   350.6    2211   363.7 2210.72   393.2  2213.4   432.5 2209.08  454.512201.542
   458.7 2201.23   468.5 2201.41   488.2 2202.42   511.1 2207.55   530.7 2226.24
   540.5  2245.6   543.8 2249.96   573.2 2276.11   589.6 2285.08     619 2307.24
   628.8  2310.9   707.4 2366.36   779.3 2419.49   870.9 2489.57   926.6 2528.19
#Mann= 3 ,-1 , 0
       0     .12       0  454.51    .045       0   468.5     .12       0
Bank Sta=454.51,468.5
XS Rating Curve= 0 ,0
Exp/Cntr=0.3,0.1

Type RM Length L Ch R = 1 ,16914   ,348.2,350,354.1
XS GIS Cut Line= 3
     2143482.184      240019.814     2143150.484      240334.114
     2142827.717      240657.996
#Sta/Elev= 30
       0 2268.54    52.2 2257.66   159.9 2232.27   182.8 2220.29   202.4 2212.74
   215.4 2209.89   277.4 2207.85   378.6 2207.89   385.2 2206.16   394.9 2199.03
   430.8 2198.94   449.5 2195.37   463.5 2195.29   464.5 2195.36   479.8 2201.64
     519 2205.87   535.3  2214.4   564.7 2235.44   587.6 2254.03   597.4 2264.67
   607.2 2281.87     617 2290.32   675.8 2330.93     715 2359.88   724.8 2364.22
   734.6 2372.71   786.8 2410.81   855.4 2457.91   884.8 2473.81   914.2 2485.41
#Mann= 3 ,-1 , 0
       0     .12       0   449.5    .045       0   464.5     .12       0
Bank Sta=449.5,464.5
XS Rating Curve= 0 ,0
Exp/Cntr=0.3,0.1

Type RM Length L Ch R = 1 ,16564   ,350.2,350,347.1
XS GIS Cut Line= 3
     2143330.141       239750.48     2142981.028       240036.99
     2142590.557      240303.157
#Sta/Elev= 30
       0 2226.59     9.8 2224.42    39.3 2224.46    98.2 2218.04   117.8 2221.47
   147.3 2221.26   166.9 2219.57   202.9 2210.86   317.4 2205.04   340.4 2206.72
   356.7 2205.33   366.5  2208.9   382.9  2208.7   392.7  2205.8   405.8 2197.14
   428.7 2195.65   444.1 2190.85   451.6 2190.38   459.1 2190.72   487.5 2192.02
   510.3 2198.94     582 2196.99   591.8 2199.51   637.4 2228.59   709.1 2278.98
   735.2 2304.42     771 2316.79   819.9 2342.78   855.8 2358.52   924.2 2377.34
#Mann= 3 ,-1 , 0
       0     .12       0   444.1    .045       0   459.1     .12       0
#XS Ineff= 2 , 0
          427.24  2201.1  508.77         2206.17
Permanent Ineff=
       F       F
Bank Sta=444.1,459.1
XS Rating Curve= 0 ,0
Exp/Cntr=0.3,0.1

Type RM Length L Ch R = 1 ,16214   ,349,350.6,349.3
XS GIS Cut Line= 3
     2143086.769      239486.827     2142742.147      239783.912
     2142396.246      240079.517
#Sta/Elev= 30
       0  2301.4    85.1 2271.92   134.2 2252.35   219.3 2227.11   284.8 2212.57
   294.6 2208.53     311 2198.01   317.5 2195.73   353.5 2193.62   396.1 2195.96
   412.4 2190.06  446.12  2185.9   451.7 2185.36   461.6 2185.97   471.4 2187.42
     491 2194.87   500.8 2196.05     599 2190.42   615.4  2191.3     635 2197.38
   687.4 2195.04   697.2 2195.89   716.9 2203.92   752.9    2224   779.1  2239.9
   811.8  2261.7     838 2276.42   860.9 2292.09   890.4 2302.92     910 2307.08
#Mann= 3 ,-1 , 0
       0     .12       0  446.12    .045       0   461.6     .12       0
#XS Ineff= 2 , 0
          390.09 2200.57  501.55         2200.81
Permanent Ineff=
       F       F
Bank Sta=446.12,461.6
XS Rating Curve= 0 ,0
Exp/Cntr=0.3,0.1

Type RM Length L Ch R = 1 ,15863.3 ,589.5,590,593.5
XS GIS Cut Line= 3
     2142885.746      239240.808     2142523.866      239512.217
     2142206.438      239858.852
#Sta/Elev= 30
       0 2365.42    13.1 2360.19    45.9 2343.58   114.7 2303.08   150.8 2291.16
   163.9  2288.7   203.2 2274.99   222.9 2266.34   249.1 2251.46     295 2229.66
   321.2 2212.59   340.9 2197.04   350.7 2191.36   370.4  2189.1   409.7 2189.24
     4362181.488   442.5 2181.39   452.4  2181.5   465.4 2181.61   478.5 2184.31
   488.2 2184.26   520.9  2188.4   543.7 2187.25   661.2 2187.55   716.7 2184.32
   772.2  2192.3   791.8 2198.17   860.4 2206.92   876.7 2211.34   922.4 2232.45
#Mann= 3 ,-1 , 0
       0     .12       0     436    .045       0   452.4     .12       0
#XS Ineff= 2 , 0
          402.48 2195.19  511.87         2194.76
Permanent Ineff=
       F       F
Bank Sta=436,452.4
XS Rating Curve= 0 ,0
Exp/Cntr=0.3,0.1

Type RM Length L Ch R = 1 ,15273.4 ,457.4,460.3,460.3
XS GIS Cut Line= 2
     2142501.275      238941.781     2141711.558      239462.426
#Sta/Elev= 30
       0 2444.13    26.2 2430.31    39.3 2420.83    55.6  2416.4    75.3 2402.98
    88.4 2396.99   121.1 2373.93   130.9 2370.44   186.6 2334.26   229.1 2302.49
   337.1 2214.75   376.4 2185.92   399.3 2176.28   428.8 2177.66     455  2170.9
   481.1 2176.16   556.4 2172.24   572.8 2172.24   589.1  2172.6   618.6 2177.01
   657.9 2175.15   700.4 2178.91   736.4 2176.57   765.9 2178.42   782.2 2181.56
   795.3 2186.68   818.2 2209.79   831.3 2218.57   883.7 2228.71   945.9 2250.94
#Mann= 3 ,-1 , 0
       0     .12       0   556.4    .045       0   572.8     .12       0
#XS Ineff= 2 , 0
          425.18 2183.45  698.66         2186.99
Permanent Ineff=
       F       F
Bank Sta=556.4,572.8
XS Rating Curve= 0 ,0
Exp/Cntr=0.3,0.1

Type RM Length L Ch R = 1 ,14813   ,357.8,368.3,375.9
XS GIS Cut Line= 3
     2142329.143      238588.598     2141945.796      238830.716
     2141547.832      239069.383
#Sta/Elev= 30
       0 2329.63    26.1  2327.7    42.4 2324.44    78.3  2311.8   114.2 2305.11
   172.9 2290.16   208.8 2279.49   221.8 2273.86   234.9 2269.86   309.9  2240.3
   394.7 2198.15     411 2185.56   430.6 2167.39   437.1 2164.52  445.022163.589
   450.1 2163.14  458.632163.589   482.8 2164.66   505.7 2169.17   561.2 2166.94
   577.6 2169.64   613.5 2168.22   636.4 2171.79   783.5  2170.3     790 2172.88
   809.6 2186.36   822.7  2193.1   865.2 2209.86     888 2217.11   917.4 2224.44
#Mann= 3 ,-1 , 0
       0     .12       0  445.02    .045       0  458.63     .12       0
Bank Sta=445.02,458.63
XS Rating Curve= 0 ,0
Exp/Cntr=0.3,0.1

Type RM Length L Ch R = 1 ,14444.8 ,333,331.7,327.3
XS GIS Cut Line= 2
     2142210.327      238471.451     2141263.103      238637.707
#Sta/Elev= 30
       0 2274.22    39.2 2254.27    68.7 2242.75   134.1 2223.14   176.6 2207.35
     229 2195.93   281.3 2180.21   300.9 2175.69   323.8 2166.67   340.2 2165.42
   353.3  2161.1   402.4 2162.66     422 2162.08   438.3 2159.37   464.5 2161.15
   499.7 2158.57     507 2157.97   513.6 2158.58   523.4 2162.69   529.9  2163.1
   667.3 2163.27   683.7  2171.1     736 2202.46   745.8 2206.84   755.6 2213.66
   775.2 2222.32     808 2234.34     857 2255.64   925.7 2272.54   961.7 2284.38
#Mann= 3 ,-1 , 0
       0     .12       0   499.7    .045       0   513.6     .12       0
#XS Ineff= 2 , 0
                          554.18         2168.38
Permanent Ineff=
       F       F
Bank Sta=499.7,513.6
XS Rating Curve= 0 ,0
Exp/Cntr=0.3,0.1

Type RM Length L Ch R = 1 ,14113   ,346.3,350,355.2
XS GIS Cut Line= 3
     2142057.008      238156.186     2141606.875      238244.845
     2141179.267      238403.012
#Sta/Elev= 30
       0 2220.62    75.4 2200.48   134.4 2186.66     154 2179.47   183.5 2165.36
   199.9 2160.22     308 2159.09   344.1 2153.92   357.2 2156.45   376.9  2157.6
   416.2  2157.1   432.6 2155.95  450.182152.261   455.5  2151.9   465.3 2152.22
   478.5 2152.83   491.6 2156.23   547.3 2195.12   553.9 2200.35   560.5  2207.1
   573.6 2229.22   576.9 2232.77   632.6 2254.44     649 2259.08     672 2263.86
   721.2  2264.8   760.5 2268.18   799.9  2275.9   881.9 2299.76   914.7 2305.69
#Mann= 3 ,-1 , 0
       0     .12       0  450.18    .045       0   465.3     .12       0
Bank Sta=450.18,465.3
XS Rating Curve= 0 ,0
Exp/Cntr=0.3,0.1

Type RM Length L Ch R = 1 ,13763   ,250.9,239.4,229
XS GIS Cut Line= 3
     2142053.502      237880.238     2141599.329      237901.119
     2141145.867      237957.595
#Sta/Elev= 30
       0 2228.34    52.3 2207.92    98.1 2193.83   147.2 2173.34   176.6 2166.78
   202.8 2152.39   209.3 2150.35   215.9 2149.78   232.2 2152.93   281.3 2152.85
   310.7 2150.16   327.1 2151.75   415.4 2153.33   431.8  2151.4   441.6 2147.03
   447.2 2146.37   451.4 2146.26   462.2 2146.35   480.8 2149.86   500.4 2148.73
   516.7 2152.36   539.5 2159.94   559.1 2169.24   604.8  2196.7   624.4 2206.43
   666.8 2230.55   699.5 2244.94     719 2252.29   794.1  2272.9   911.6 2314.41
#Mann= 3 ,-1 , 0
       0     .12       0   447.2    .045       0   462.2     .12       0
#XS Ineff= 2 , 0
                          486.07         2157.03
Permanent Ineff=
       F       F
Bank Sta=447.2,462.2
XS Rating Curve= 0 ,0
Exp/Cntr=0.3,0.1

Type RM Length L Ch R = 1 ,13523.6 ,461.1,460,459.4
XS GIS Cut Line= 2
      2141980.63      237392.972      2141129.66      237931.118
#Sta/Elev= 30
       0 2296.72    72.2 2276.15   111.5 2260.46   147.6 2243.35   239.4 2188.75
   249.2  2181.1     282 2151.26   295.2 2144.72   301.7 2143.69   350.9 2146.35
     364 2145.26   393.6 2147.42   413.2 2143.55   452.6 2148.41     469 2148.73
     492 2148.24  523.282143.136     528  2142.9   537.9 2143.06   570.7 2151.74
   606.7 2151.37   629.7 2148.13   655.9 2150.06   682.2 2166.16   734.6 2206.54
   770.7 2229.65   793.7 2240.61   888.8 2275.54     938 2292.07  1006.8 2321.76
#Mann= 3 ,-1 , 0
       0     .12       0  523.28    .045       0   537.9     .12       0
Bank Sta=523.28,537.9
XS Rating Curve= 0 ,0
Exp/Cntr=0.3,0.1

Type RM Length L Ch R = 1 ,13063.6 ,357.3,350.4,338.8
XS GIS Cut Line= 3
     2141831.382      236986.903      2141475.83      237251.292
     2141033.885      237530.124
#Sta/Elev= 30
       0 2322.44    39.1 2309.11     114 2276.36   156.4  2259.7   211.8 2232.38
   293.2 2195.32   322.5  2185.9   368.2 2176.82   384.4 2171.51   400.7 2160.68
   420.3 2138.61  434.552134.796   443.1 2134.34   449.6 2134.76   475.7 2138.87
   495.3 2138.47   511.7 2140.61   560.6  2140.7   609.6 2136.38   622.7 2137.21
     639 2141.24     688  2138.5   733.8 2143.81   756.6 2156.98   795.8 2185.09
   799.1 2188.12   805.6 2198.04   812.1 2204.27   923.2 2274.84   965.6 2303.64
#Mann= 3 ,-1 , 0
       0     .12       0  434.55    .045       0   449.6     .12       0
#XS Ineff= 2 , 0
                          557.28         2146.45
Permanent Ineff=
       F       F
Bank Sta=434.55,449.6
XS Rating Curve= 0 ,0
Exp/Cntr=0.3,0.1

Type RM Length L Ch R = 1 ,12713.2 ,347.2,348.6,351.2
XS GIS Cut Line= 3
     2141453.003      236687.319     2141189.983      237057.247
     2140956.855      237467.944
#Sta/Elev= 30
       0 2248.88    16.3  2240.2    35.9 2231.79   137.2  2195.1   163.3 2183.05
   202.5 2168.94   235.1 2159.69   300.4 2146.63   333.1 2138.13     369 2136.78
   408.2 2137.95   414.7 2136.89   421.2 2133.06     431 2129.98   453.9 2129.75
   463.7 2129.59  468.242129.763   496.5 2134.15   535.9 2134.12   552.3 2132.39
   578.5 2133.78   611.3  2131.3   617.9 2133.31   634.3 2143.85     654 2158.95
   683.5 2182.68   699.9  2199.4   726.1 2217.71   870.4 2301.75   926.2  2332.9
#Mann= 3 ,-1 , 0
       0     .12       0   453.9    .045       0  468.24     .12       0
#XS Ineff= 2 , 0
                          578.95         2140.54
Permanent Ineff=
       F       F
Bank Sta=453.9,468.24
XS Rating Curve= 0 ,0
Exp/Cntr=0.3,0.1

Type RM Length L Ch R = 1 ,12364.5 ,389.6,394.9,399.4
XS GIS Cut Line= 3
      2141152.12      236546.689     2140881.924      236912.821
     2140607.513       237275.75
#Sta/Elev= 30
       0 2199.09    22.9 2189.63      36 2186.82   101.5 2163.11   111.3 2161.75
     144 2152.66     180 2141.12   225.9 2131.57   242.2    2130   314.3 2129.01
   340.5 2133.38   363.4 2127.99   379.7 2129.25   412.5 2127.12   428.8 2124.96
   435.4 2121.71   445.2 2121.15   458.3 2120.95  459.95 2121.13   471.4 2124.86
   484.5 2140.17   497.6 2152.69     514 2166.89   530.3 2178.41   602.3  2224.2
     694 2278.26   746.4 2307.07   798.7 2332.52   857.7  2359.1     910 2380.27
#Mann= 3 ,-1 , 0
       0     .12       0   445.2    .045       0  459.95     .12       0
#XS Ineff= 2 , 0
          381.17 2135.08
Permanent Ineff=
       F       F
Bank Sta=445.2,459.95
XS Rating Curve= 0 ,0
Exp/Cntr=0.3,0.1

Type RM Length L Ch R = 1 ,11969.6 ,320.9,305.1,289.7
XS GIS Cut Line= 4
     2140879.462      236414.427      2140530.56      236716.452
     2140379.234      236856.393     2140374.482      237048.004
#Sta/Elev= 30
       0 2167.49     9.8 2168.85    22.9 2167.54    49.1 2170.53    88.4 2170.14
   134.2 2161.42   176.7 2154.82   219.3 2151.54   238.9  2148.8   248.7 2145.46
   265.1  2135.2   284.7 2125.13   291.3 2122.83   330.6 2120.31   353.5 2120.17
   369.8 2117.59   389.5 2118.18  408.03 2114.75   422.2 2114.58   425.5 2114.73
   441.8 2120.04   451.6 2121.98   510.5 2120.02     540 2123.43   602.2 2120.73
   670.8 2128.64   693.6 2134.36   735.8 2149.33   800.8 2184.13   859.2 2213.93
#Mann= 3 ,-1 , 0
       0     .12       0  408.03    .045       0   425.5     .12       0
#XS Ineff= 2 , 0
          355.01 2125.74  459.24         2127.57
Permanent Ineff=
       F       F
Bank Sta=408.03,425.5
XS Rating Curve= 0 ,0
Exp/Cntr=0.3,0.1

Type RM Length L Ch R = 1 ,11664.5 ,353.4,350,345.9
XS GIS Cut Line= 3
      2140357.48      236136.253     2140288.053      236585.881
     2140205.145      237033.516
#Sta/Elev= 30
       0 2320.17    16.4 2304.32      36 2290.16    49.1 2277.01    65.5 2276.04
    68.7 2274.24    78.6 2263.48    91.6 2252.44   163.6  2205.8   245.5 2159.43
   291.3 2138.02   301.1 2135.91   327.3 2119.36   369.9 2115.61   399.3  2115.8
     432 2108.78   447.5 2108.03   462.5 2107.99   468.1 2107.95   504.1 2117.86
   517.2 2118.77   576.1 2120.08   631.8 2116.02   674.4 2119.12   743.2 2118.95
   756.3 2120.58   792.3 2139.59     884 2201.14   893.8 2211.93   910.2 2222.35
#Mann= 3 ,-1 , 0
       0     .12       0   447.5    .045       0   462.5     .12       0
Bank Sta=447.5,462.5
XS Rating Curve= 0 ,0
Exp/Cntr=0.3,0.1

Type RM Length L Ch R = 1 ,11314.5 ,348.7,350,351.7
XS GIS Cut Line= 3
     2139940.851      236092.142     2139940.851      236547.142
     2139940.851      237002.142
#Sta/Elev= 30
       0 2263.26    26.2 2245.69    55.6 2244.93    78.6 2228.72    88.4 2224.86
   137.5 2212.72   153.8 2205.51   166.9 2204.84   189.9 2194.78   235.7 2164.55
   271.7 2131.41   304.4 2109.87   317.5  2106.8   337.2 2109.62   392.8 2107.94
   415.7 2110.84   428.8  2109.5   435.4  2105.2   445.2 2103.58     455 2103.31
   461.6 2103.57   533.6 2107.45   553.2  2113.2   582.7 2110.76   612.1 2112.88
   667.8 2111.83   710.3 2118.92   746.3 2131.98   798.7 2156.46     910 2221.39
#Mann= 3 ,-1 , 0
       0     .12       0   445.2    .045       0   461.6     .12       0
#XS Ineff= 2 , 0
          414.86 2116.72
Permanent Ineff=
       F       F
Bank Sta=445.2,461.6
XS Rating Curve= 0 ,0
Exp/Cntr=0.3,0.1

Type RM Length L Ch R = 1 ,10964.5 ,343.6,350.8,356.8
XS GIS Cut Line= 3
     2139619.897       236120.35     2139596.186      236584.525
     2139558.656      237036.223
#Sta/Elev= 30
       0    2250     9.8 2239.55    29.5 2237.72    65.5 2210.34    75.3 2201.52
    91.6 2195.52   153.8 2147.61   193.1 2114.97   206.2  2105.7     216 2101.07
   225.8 2099.36   245.5 2101.54   278.2 2101.06   320.8 2105.13   350.2 2103.26
     396 2104.76  460.172097.569     468  2097.4   474.6 2097.55   494.1 2104.97
   523.5  2104.6   536.5  2106.8   611.5  2105.7   653.9 2109.26   670.2 2112.17
   689.8 2120.68     768 2169.85   797.4 2185.08   856.1 2219.42     918 2253.23
#Mann= 3 ,-1 , 0
       0     .12       0  460.17    .045       0   474.6     .12       0
#XS Ineff= 2 , 0
          397.32 2110.41
Permanent Ineff=
       F       F
Bank Sta=460.17,474.6
XS Rating Curve= 0 ,0
Exp/Cntr=0.3,0.1

Type RM Length L Ch R = 1 ,10613.7 ,349.7,351.4,351.6
XS GIS Cut Line= 3
     2139421.893      236058.291     2139262.043      236484.304
     2139099.039      236909.101
#Sta/Elev= 30
       0 2228.44     9.8 2226.69      36 2212.12    45.8 2210.09   114.6  2180.5
   127.7 2173.52   137.5 2172.26   160.4 2159.94   212.8 2139.96   222.6 2134.24
   258.6 2103.37   268.4 2097.32     275 2095.94   314.3 2095.22   343.7 2097.37
   369.9 2097.32   386.3 2095.39     419 2097.29   435.4 2090.93   445.2 2090.76
   451.7 2090.94   487.8 2093.39   507.4  2097.7   592.5  2102.3     622 2109.12
   671.1 2115.05   703.8 2126.71   743.1 2137.48   759.4 2144.02     910 2220.04
#Mann= 3 ,-1 , 0
       0     .12       0   435.4    .045       0   451.7     .12       0
#XS Ineff= 2 , 0
          416.92 2101.08
Permanent Ineff=
       F       F
Bank Sta=435.4,451.7
XS Rating Curve= 0 ,0
Exp/Cntr=0.3,0.1

Type RM Length L Ch R = 1 ,10262.3 ,353.5,354.2,355.5
XS GIS Cut Line= 3
     2139114.657       235965.35     2138928.277      236381.291
     2138760.602      236804.119
#Sta/Elev= 30
       0 2163.36      23 2151.25    39.4 2147.23    78.7 2133.01   131.2 2109.45
     200 2094.89   219.7 2094.97   232.8 2090.63   239.4 2089.83   278.7  2091.7
   347.6 2089.87   403.3  2091.3   416.4 2090.65   419.7 2089.23     423 2085.39
   426.3 2084.45     446 2083.01   455.8 2082.92  460.582082.994     482 2084.47
   501.6 2089.21   537.6 2089.56     554 2088.47   580.1  2094.9   632.5 2096.53
   655.4 2098.72   724.1 2111.06   769.9 2125.36   858.3 2163.92   910.6 2185.31
#Mann= 3 ,-1 , 0
       0     .12       0     446    .045       0  460.58     .12       0
#XS Ineff= 2 , 0
          398.35 2095.61  524.25         2093.58
Permanent Ineff=
       F       F
Bank Sta=446,460.58
XS Rating Curve= 0 ,0
Exp/Cntr=0.3,0.1

Type RM Length L Ch R = 1 ,9908.2  ,542.4,546,546.8
XS GIS Cut Line= 2
     2138794.049      235851.246     2138411.221      236654.089
#Sta/Elev= 30
       0 2129.21    19.6 2118.04      36 2114.17    68.7 2095.46    88.3 2088.44
   117.7 2087.58   212.6 2090.92   255.1 2089.31   313.9 2090.94   340.1 2088.48
   353.2 2085.85   369.5 2086.19   385.9 2084.43   408.8 2079.91   431.6 2080.81
     448 2079.42   451.3 2079.08     461  2079.4   477.4 2083.55   490.5 2084.83
   595.1 2082.23   611.5 2083.93   621.3 2086.38   637.6 2093.28   670.4 2099.13
   706.3 2107.61   735.8 2116.88   771.7 2131.82     811 2152.54   889.4 2198.47
#Mann= 3 ,-1 , 0
       0     .12       0     448    .045       0     461     .12       0
#XS Ineff= 2 , 0
          381.84 2089.09
Permanent Ineff=
       F       F
Bank Sta=448,461
XS Rating Curve= 0 ,0
Exp/Cntr=0.3,0.1

Type RM Length L Ch R = 1 ,9362.2  ,494.9,498.7,503
XS GIS Cut Line= 2
     2138392.993      235732.596     2137983.914      236500.438
#Sta/Elev= 30
       0 2096.12    32.7  2082.3    45.8 2080.39    88.3  2081.2   107.9 2078.69
     157 2085.18   199.5 2085.67     229 2077.39   297.6  2078.7   327.1  2077.1
   369.6 2080.15   405.6  2077.9   474.3 2081.23   546.2 2075.44   562.6 2077.82
   582.2 2077.95   618.2 2075.17   632.7 2071.18   644.3 2070.78   647.7  2071.3
   657.4 2077.91   670.5 2093.56   699.9 2119.61   722.8 2146.49   755.5 2175.63
   765.4 2182.19     785 2190.23   817.7 2218.09   847.1 2237.49     870 2254.98
#Mann= 3 ,-1 , 0
       0     .12       0   632.7    .045       0   647.7     .12       0
#XS Ineff= 2 , 0
          475.75  2089.7
Permanent Ineff=
       F       F
Bank Sta=632.7,647.7
XS Rating Curve= 0 ,0
Exp/Cntr=0.3,0.1

Type RM Length L Ch R = 1 ,8863.5  ,354.9,350.2,344.4
XS GIS Cut Line= 3
     2138016.906      235591.866     2137744.018      235956.598
     2137434.761      236291.634
#Sta/Elev= 30
       0 2076.39    85.2 2074.53   111.4 2070.32   150.8 2071.46   180.2  2068.6
   206.5 2072.83   265.4 2069.75   288.4 2072.09   353.9  2071.9   376.9  2068.7
   416.2 2070.12   435.9 2065.84   439.1 2065.73   452.2 2065.81     508 2071.23
   524.4 2082.59     531 2095.95   537.5 2104.08   557.2 2121.26   570.3 2129.89
   622.8  2144.3     649  2154.5   668.7 2156.99   734.3 2182.39   786.8 2207.47
   806.5 2214.53   829.5 2218.31   855.7 2215.75     882 2208.84   911.5  2194.1
#Mann= 3 ,-1 , 0
       0     .12       0   435.9    .045       0   452.2     .12       0
#XS Ineff= 2 , 0
          300.31  2077.3
Permanent Ineff=
       F       F
Bank Sta=435.9,452.2
XS Rating Curve= 0 ,0
Exp/Cntr=0.3,0.1
